--- BCKLERN.prj (project) ---

Proj Title=BCKLERN
Current Plan=p01
Default Exp/Contr=0,0
English Units
Geom File=g01
Flow File=f01
Plan File=p01
BEGIN DESCRIPTION:
----------MODEL BY WOOD PLC 2022----------
AFH study
Randolph County, WV
HEC-RAS Version: RAS 6.2
Vertical Datum: NAVD88
Projection: NAD 1983 StatePlane West Virginia S FIPS 4702 (US Feet)
Terrain: 1-meter LIDAR (FEMA Region III 3DEP collected 2016-2018)
Land Use: 2019 NLCD
Hydrologic Method:
WV SIR2010-5033 regression equations
Additional Model Notes:
None
END DESCRIPTION:
DSS Export Rating Curves= 0
DSS Export Rating Curve Sorted= 0
DSS Export Volume Flow Curves= 0
DXF OffsetX= 0
DXF OffsetY= 0
DXF ScaleX= 0
DXF ScaleY= 0

--- BCKLERN.p01 (plan) ---

Plan Title=Floodplain
Program Version=6.20
Short Identifier=Floodplain
Geom File=g01
Flow File=f01
Subcritical Flow
K Sum by GR= 0
Std Step Tol= 0.01
Critical Tol= 0.01
Num of Std Step Trials= 20
Max Error Tol= 0.3
Flow Tol Ratio= 0.001
Split Flow NTrial= 30
Split Flow Tol= 0.02
Split Flow Ratio= 0.02
Log Output Level= 0
Friction Slope Method= 1
Unsteady Friction Slope Method= 2
Unsteady Bridges Friction Slope Method= 1
Parabolic Critical Depth
Global Vel Dist= 0 , 0 , 0
Global Log Level= 0
CheckData=True
Encroach Param=-1 ,0,0, 0
Mapping Interval=1HOUR
Computation Time Step Use Courant=        0
Computation Time Step Use Time Series=    0
Computation Time Step Count To Double=0
Computation Time Step Max Doubling=0
Computation Time Step Max Halving=0
Computation Time Step Residence Courant=0
Run HTab= 0
Run UNet= 0
Run Sediment= 0
Run PostProcess= 0
Run WQNet= 0
Run RASMapper=-1
UNET Theta= 0
UNET Theta Warmup= 0
UNET ZTol= 0
UNET ZSATol= 0
UNET MxIter= 0
UNET Max Iter WO Improvement= 0
UNET MaxInSteps= 0
UNET DtIC= 0
UNET DtMin= 0
UNET MaxCRTS= 0
UNET WFStab= 0
UNET SFStab= 0
UNET WFX= 1
UNET SFX= 1
UNET Gravity=32.174
UNET 1D Methodology=Finite Difference
UNET DSS MLevel= 1
UNET Pardiso=0
UNET DZMax Abort= 0
UNET Use Existing IB Tables= 0
UNET Froude Reduction=False
UNET Froude Limit= 0
UNET Froude Power= 0
UNET D1 Cores= 0
UNET WindReference=Eulerian
UNET WindDragFormulation=Hsu (1988)
UNET D2 Coriolis=0
UNET D2 Cores= 0
UNET D2 Theta= 1
UNET D2 Theta Warmup= 1
UNET D2 Z Tol= 0.01
UNET D2 Volume Tol= 0.01
UNET D2 Max Iterations= 20
UNET D2 Equation= 0
UNET D2 RampUpFraction=0.1
UNET D2 TimeSlices= 1
UNET D2 Turbulence Formulation=Non-Conservative (original)
UNET D2 Eddy Viscosity=0.3
UNET D2 Transverse Eddy Viscosity=0.1
UNET D2 Smagorinsky Mixing=0
UNET D2 BCVolumeCheck=0
UNET D2 Cores=0
UNET D2 SolverType=PARDISO (Direct)
UNET D2 Minimum Iterations= 2147483647
UNET D2 Maximum Iterations= 2147483647
UNET D2 Restart Number= 10
UNET D2 Relaxation Coeff=1.3
UNET D2 SOR Precondition Iterations= 10
UNET D2 ILUT Maximum Fill= 8
UNET D2 ILUT Tolerance=1E-08
UNET D1D2 MaxIter= 0
UNET D1D2 ZTol=0.01
UNET D1D2 QTol=0.1
UNET D1D2 MinQTol=1
Write IC File= 0
Write IC File at Fixed DateTime=0
Write IC File at Sim End=0
Echo Input=False
Echo Parameters=False
Echo Output=False
Write Detailed= 0
HDF Write Warmup=0
HDF Write Time Slices=0
HDF Flush=0
HDF Compression= 1
HDF Chunk Size= 1
HDF Spatial Parts= 1
HDF Use Max Rows=0
HDF Fixed Rows= 1
Calibration Method= 0
Calibration Iterations= 20
Calibration Max Change=0.05
Calibration Tolerance=0.2
Calibration Maximum=1.5
Calibration Minimum=0.5
Calibration Optimization Method= 1
WQ AD Non Conservative
WQ ULTIMATE=-1
WQ Max Comp Step=1HOUR
WQ Output Interval=15MIN
WQ Output Selected Increments= 0
WQ Output face flow=0
WQ Output face velocity=0
WQ Output face area=0
WQ Output face dispersion=0
WQ Output cell volume=0
WQ Output cell surface area=0
WQ Output cell continuity=0
WQ Output cumulative cell continuity=0
WQ Output face conc=0
WQ Output face dconc_dx=0
WQ Output face courant=0
WQ Output face peclet=0
WQ Output face adv mass=0
WQ Output face disp mass=0
WQ Output cell mass=0
WQ Output cell source sink temp=0
WQ Output nsm pathways=0
WQ Output nsm derived pathways=0
WQ Create Restart=0
WQ Fixed Restart=0
WQ System Summary=0
WQ Write To DSS=0
Sorting and Armoring Iterations= 10
XS Update Threshold= 0.02
Bed Roughness Predictor= 0
Hydraulics Update Threshold= 0.02
Energy Slope Method= 1
Volume Change Method= 1
Sediment Retention Method= 0
Sediment TS Multiplier= 1
Warm Up Method= 0
XS Weighting Method= 0
Number of US Weighted Cross Sections= 1
Number of DS Weighted Cross Sections= 1
Upstream XS Weight=0
Main XS Weight=1
Downstream XS Weight=0
Number of DS XS's Weighted with US Boundary= 1
Upstream Boundary Weight= 1
Weight of XSs Associated with US Boundary= 0
Number of US XS's Weighted with DS Boundary= 1
Downstream Boundary Weight= 0.5
Weight of XSs Associated with DS Boundary= 0.5
Percentile Method= 0
Sediment Output Level= 3
Mass or Volume Output= 0
Output Increment Type= 1
Profile and TS Output Increment= 1
Transport Output Increment 1
XS Output Flag= 0
XS Output Increment= 10
Read HDF5 Sediment Hotstart= 0
Sediment Hotstart Type= 0
Write Gradation File= 0
Read Gradation Hotstart= 0
Write HDF5 File= 1
Write Binary Output= 1
Write DSS Sediment File= 0
DSS Sediment Output Type= 1
SV Curve= 0
Specific Gage Flag= 0
Subcell Erosion Methods= 0
Subcell Deposition Methods= 0
Advection Scheme= 1
Matrix Solver= 0
Implicit Weighting Factor= 1
Maximum Outer Loop Convergence Iterations= 5
Convergence Maximum Absolute= 0.001
Convergence RMSE= 0.0001
Grain Fractions Max Abs Error= 0.001
Max Subgrid Regions= 1
Max Subgrid Length Scale= 3.402823E+38
Initial Layer Thickness= 3.402823E+38
Min Layer Thickness= 3.402823E+38
Max Layer Thickness= 3.402823E+38
Number of Layers= 5

--- BCKLERN.f01 (steady flow) ---

Flow Title=Flow
Program Version=6.20
Number of Profiles= 1
Profile Names=P100yr
River Rch & RM=BCKLERN,Main            ,5288
     371
River Rch & RM=BCKLERN,Main            ,4021
     413
River Rch & RM=BCKLERN,Main            ,3115
     468
Boundary for River Rch & Prof#=BCKLERN,Main            , 1
Up Type= 0
Dn Type= 3
Dn Slope=0.04379
DSS Import GetInterval= 0
DSS Import GetPeak= 0
DSS Import FillOption= 0

--- BCKLERN.g01 (geometry) ---

Geom Title=Geometry
Program Version=6.20

River Reach=BCKLERN         ,Main
Reach XY= 30
2334286.66296653702700.422949795     2334312.161      702617.699
     2334289.405      702432.255     2334417.293      702025.882
     2334299.932      701757.479     2334299.585      701688.729
2334386.65449723701465.184460314     2334449.932      701420.326
2334601.16006025701207.126286168     2334648.283      701087.427
2334820.06507531701039.405015061     2334921.286      700648.191
     2334870.071       700503.66 2334937.3625658700426.004131605
     2334987.692      700286.212     2335081.443      700208.521
2335163.44061191699905.809782901     2335161.521      699776.374
     2335093.812      699630.1932335081.71270333 699471.80629667
     2335111.694      699338.657     2335087.714      699193.391
     2335139.363      698858.105     2335098.565      698785.839
     2334993.906      698736.302     2334969.254      698521.719
     2334995.643      698417.552 2335106.2716892      698281.311
 2335143.7877558698184.367844601     2335268.891      698108.095

Type RM Length L Ch R = 1 ,5288    ,96.3,93.8,93.2
XS GIS Cut Line= 3
2334559.96623606702737.8092485682334220.62807936702680.478252768
2334000.91935693702738.508612828
#Sta/Elev= 30
       0 2607.31    52.7 2585.68      89  2567.6   105.3 2562.77   117.4 2556.45
   128.8 2553.46   149.9 2544.69   182.3 2534.63   190.5    2530   198.6 2528.82
   214.8 2517.61   222.9 2506.47   243.2 2488.59   251.3 2486.83   263.5 2487.68
  273.242483.881   279.7 2483.09   284.9 2483.91   287.8 2485.27   295.9 2494.16
   324.3 2511.13   369.4 2521.42   409.5 2536.82   423.2 2539.66   443.3 2546.89
   489.4 2568.39   522.5 2580.91   534.9 2588.94     548 2592.18   571.4 2605.15
#Mann= 3 ,-1,0
       0      .1       0  273.24    .045       0   284.9      .1       0
Bank Sta=273.24,284.9
XS Rating Curve= 0 ,0
Exp/Cntr(USF)=0,0
Exp/Cntr=0.3,0.1

Type RM Length L Ch R = 1 ,5194    ,99.6,99,98.8
XS GIS Cut Line= 3
 2334590.1643309702648.410153967 2334345.0913444702600.466153811
2334004.43162311702626.234012297
#Sta/Elev= 30
       0 2617.19    10.2 2610.51    46.9 2592.24    75.4 2580.07    87.6 2572.55
   120.2 2556.24     161 2539.22   173.2 2536.84   185.4 2532.62   193.6 2528.21
   202.2 2526.59   234.3  2511.1   250.6 2500.94   266.7 2484.59   274.7 2479.82
   282.7 2479.37287.24522479.845   310.7 2482.92   342.9  2494.2     367  2499.5
   399.1 2508.75   415.1 2515.79   439.2 2523.17   459.2 2526.01     475 2531.27
     516 2540.59   539.5 2548.88   563.5 2553.51   575.7 2562.27   591.4 2567.17
#Mann= 3 ,-1,0
       0      .1       0   274.7    .045       0287.2452      .1       0
Bank Sta=274.7,287.2452
XS Rating Curve= 0 ,0
Exp/Cntr(USF)=0,0
Exp/Cntr=0.3,0.1

Type RM Length L Ch R = 1 ,5095    ,137.2,139.7,145.1
XS GIS Cut Line= 4
2334609.45131935702576.3386310482334310.09823611702503.861865008
2334256.18027575702510.8534557722334027.04024136702486.599897988
#Sta/Elev= 30
       0 2611.63      26 2600.55    42.5 2591.61    66.6 2580.35    76.6 2577.38
    91.9 2569.09   100.1 2566.16   136.2 2548.47   174.2 2532.39   190.6 2527.06
   195.8  2524.3   207.1 2521.63   256.5 2499.66   285.3 2486.44   289.4 2483.78
   293.5 2479.38   297.6 2477.24   309.9 2477.46  318.34 2475.36     322 2474.22
   328.82475.377   349.4 2487.72   362.4 2497.38   394.6 2510.58   410.6 2520.43
   426.7 2528.95   462.9 2539.39   523.3 2548.61   559.5 2566.38   592.8 2578.39
#Mann= 3 ,-1,0
       0      .1       0  318.34    .045       0   328.8      .1       0
Bank Sta=318.34,328.8
XS Rating Curve= 0 ,0
Exp/Cntr(USF)=0,0
Exp/Cntr=0.3,0.1

Type RM Length L Ch R = 1 ,4956    ,110,108.1,104.5
XS GIS Cut Line= 4
2334630.82344001702480.0301644152334358.62227936702397.217641995
2334297.41302365702361.2121974642334090.02166316702331.687732949
#Sta/Elev= 30
       0 2599.74    35.8 2586.55      51 2578.73    61.3 2575.29    86.4 2560.22
   135.8 2536.84   149.1 2532.71   161.6 2526.63     174 2523.22     216 2508.12
   224.4 2504.02   236.9 2502.07   253.6 2496.82   286.3 2480.85   305.9 2477.35
   315.2 2469.62   327.2 2466.01   338.4 2465.48  340.51 2465.99   355.8 2470.32
   368.9 2476.15   432.3 2519.81   441.8 2523.16   461.8 2533.36     478 2539.25
   510.3 2545.67   522.4 2550.18   534.6 2547.27   538.6 2547.58     565 2557.27
#Mann= 3 ,-1,0
       0      .1       0   327.2    .045       0  340.51      .1       0
Bank Sta=327.2,340.51
XS Rating Curve= 0 ,0
Exp/Cntr(USF)=0,0
Exp/Cntr=0.3,0.1

Type RM Length L Ch R = 1 ,4847    ,70.6,71.7,73.3
XS GIS Cut Line= 4
2334628.66311334702453.3861354622334609.22017329702409.459493135
2334390.30707054702275.5192394822334106.58416764702240.233903842
#Sta/Elev= 30
       0 2589.47    22.1 2581.36      43 2568.99      49 2563.97    82.1 2551.59
   105.5 2538.13   153.7 2517.75   199.3 2492.19   218.1 2486.89   255.6 2486.83
   274.3 2483.64   306.8 2474.75   314.9 2470.23   326.6  2465.7     335 2459.98
   343.1 2458.63   347.1 2458.26   356.82458.658   367.3 2463.27   375.3 2470.67
   387.4 2479.57   411.6 2489.25   431.8 2499.74   443.9 2504.66   484.3 2526.16
   496.3 2528.74   508.4 2536.15   524.5 2542.54   544.6 2548.83   590.6 2559.61
#Mann= 3 ,-1,0
       0      .1       0   343.1    .045       0   356.8      .1       0
Bank Sta=343.1,356.8
XS Rating Curve= 0 ,0
Exp/Cntr(USF)=0,0
Exp/Cntr=0.3,0.1

Type RM Length L Ch R = 1 ,4776    ,129.8,128.4,127.1
XS GIS Cut Line= 4
 2334625.3372129702395.1709240042334620.02180665702287.040981731
2334226.12224348702153.8208369682334108.42052538702197.680006895
#Sta/Elev= 30
       0 2556.47      26 2543.23      34 2537.95    50.1 2531.72    70.1 2520.91
    79.4  2514.4    90.1 2504.41   108.3 2492.87   146.1 2491.87     164 2489.78
   196.8 2490.01   222.1 2485.28     239 2485.51   281.2 2477.94   293.9 2478.15
   310.8 2475.46   327.7 2468.05   336.1 2466.68   344.6 2461.21   349.4  2459.3
  371.172455.231   377.8 2454.66   384.1 2455.23   406.2 2463.59   425.1 2473.92
   459.9  2487.2   488.1 2496.38   553.1 2514.47   602.8 2536.12   649.7 2551.62
#Mann= 3 ,-1,0
       0      .1       0  371.17    .045       0   384.1      .1       0
Bank Sta=371.17,384.1
XS Rating Curve= 0 ,0
Exp/Cntr(USF)=0,0
Exp/Cntr=0.3,0.1

Type RM Length L Ch R = 1 ,4647    ,94.3,92.8,91.2
XS GIS Cut Line= 4
2334642.01057232702068.6560517592334428.43445497702083.516934379
2334269.32877692702064.5273345332334107.66835417702129.807442429
#Sta/Elev= 30
       0 2554.52    29.9 2542.19    43.4 2537.41      58 2534.67      82 2528.08
   110.1 2516.28   134.2 2501.08   166.2 2482.42   174.3 2478.92   198.3 2466.06
   210.3 2457.97   218.4 2451.73   226.4  2447.3   230.5 2446.22  239.592447.315
   262.7 2455.41   278.8 2457.46   282.8 2459.57   290.9  2462.1   323.1  2474.6
   339.2 2479.37   353.5 2482.28   374.3 2484.91   414.4 2492.72   427.3 2494.37
   470.5 2507.45   483.3 2509.47   500.7 2513.62   523.2 2522.22   548.7  2529.6
#Mann= 3 ,-1,0
       0      .1       0   226.4    .045       0  239.59      .1       0
Bank Sta=226.4,239.59
XS Rating Curve= 0 ,0
Exp/Cntr(USF)=0,0
Exp/Cntr=0.3,0.1

Type RM Length L Ch R = 1 ,4555    ,86.8,85.6,83.8
XS GIS Cut Line= 3
2334630.82297692701980.2997802172334433.35574414701985.402291837
2334121.65869882702047.727411308
#Sta/Elev= 30
       0 2559.26    34.7 2543.63    42.7 2541.69    54.7 2536.88    66.7 2534.28
    94.7 2524.62   114.7 2514.54   134.7 2501.63   142.7 2495.29     162 2483.06
   178.7 2469.61   186.7 2465.72   198.7 2456.33   206.9 2445.86  213.362442.092
   219.1  2441.2   222.1 2442.06   259.9 2454.85   276.2  2457.9   288.5 2461.69
   300.7 2462.13   325.2 2468.31   342.1 2470.39   372.7  2477.3   382.3 2480.34
   402.3 2484.12   412.5  2487.3   435.3 2491.66   459.4 2499.15   515.4  2520.1
#Mann= 3 ,-1,0
       0      .1       0  213.36    .045       0   222.1      .1       0
Bank Sta=213.36,222.1
XS Rating Curve= 0 ,0
Exp/Cntr(USF)=0,0
Exp/Cntr=0.3,0.1

Type RM Length L Ch R = 1 ,4469    ,70.8,71.2,71.5
XS GIS Cut Line= 4
2334625.06256888701903.9430519272334406.14946614701895.301745239
2334228.28257016 702002.597969942334122.42656324702019.160474424
#Sta/Elev= 30
       0 2553.54    36.9 2539.83    52.9  2535.4    64.7 2533.81    92.1 2526.27
     125 2509.64     137 2502.26     149  2493.3     169 2481.42     181  2472.7
   202.3 2459.32   213.1 2451.02   222.7 2441.03   230.7 2438.57   248.1 2441.02
   256.9 2438.75   261.4 2438.23   265.6 2438.77   272.8 2441.38   277.4  2445.2
   283.1 2448.32   319.5 2459.53   333.5 2459.53   342.8 2462.99   370.9 2469.03
   422.3 2477.29     431  2481.5   464.2 2492.55   491.7 2500.09     534 2516.18
#Mann= 3 ,-1,0
       0      .1       0   256.9    .045       0   265.6      .1       0
Bank Sta=256.9,265.6
XS Rating Curve= 0 ,0
Exp/Cntr(USF)=0,0
Exp/Cntr=0.3,0.1

Type RM Length L Ch R = 1 ,4398    ,60,56.5,54.9
XS GIS Cut Line= 3
2334609.94028218701854.2555384752334383.10598164701840.573469553
2334122.42656324701921.225665301
#Sta/Elev= 30
       0 2542.84    37.8 2531.67    49.9 2530.02    73.9 2524.05     114 2507.56
     134 2497.47   198.1 2460.99   218.2 2446.32   230.3 2439.43   242.9 2436.66
   242.9 2436.65     249 2436.21   258.9 2436.66   263.8 2438.09   272.2 2438.25
   305.7 2443.76   318.2 2444.15   330.8 2447.33   338.8 2450.31   355.9 2454.18
   385.2 2460.13   431.3 2467.64   439.7  2469.8   443.9 2471.08   452.2 2476.99
   460.6 2480.48     469 2486.32   481.5 2493.47   494.1 2498.78   500.1 2502.47
#Mann= 3 ,-1,0
       0      .1       0   242.9    .045       0   258.9      .1       0
Bank Sta=242.9,258.9
XS Rating Curve= 0 ,0
Exp/Cntr(USF)=0,0
Exp/Cntr=0.3,0.1

Type RM Length L Ch R = 1 ,4341    ,60.7,64.9,67.6
XS GIS Cut Line= 4
 2334598.3012305 701805.017511842334338.60324323701793.873250002
2334294.31772015701822.9795809892334117.26849157701858.305569745
#Sta/Elev= 30
       0 2532.78    18.1 2528.78    30.2 2526.97    56.8  2520.3   118.2 2498.82
   134.2 2490.53   142.3 2488.01   158.3 2477.61   178.5 2466.51   211.6 2450.38
   216.9 2446.65   222.3 2441.36   226.3 2438.74   236.1 2437.44   246.4 2434.09
   250.4 2434.08   258.4 2436.31   261.2 2436.21  269.98 2432.72   272.4 2431.84
   277.2 2432.74   286.8 2437.14   305.9 2441.51   327.4 2444.12   339.6 2449.76
   388.5 2459.94   426.4 2470.95   457.9 2481.24   478.3 2490.74   493.5 2499.33
#Mann= 3 ,-1,0
       0      .1       0  269.98    .045       0   277.2      .1       0
Bank Sta=269.98,277.2
XS Rating Curve= 0 ,0
Exp/Cntr(USF)=0,0
Exp/Cntr=0.3,0.1

Type RM Length L Ch R = 1 ,4276    ,77.1,84.9,88.6
XS GIS Cut Line= 3
2334606.33973773701774.3234516172334385.26630831701726.796264837
2334103.70373208701783.684867195
#Sta/Elev= 30
       0  2530.6      23 2524.93      39 2522.94    51.3 2518.94    63.6 2516.48
   127.4 2494.77   147.3 2485.34   190.4  2461.8   219.1 2450.15   227.2 2443.65
   231.3 2442.39   239.5 2442.52   243.6 2441.71   251.7 2436.28     264 2430.86
   272.1 2426.21   284.4 2423.87   293.6 2419.14   296.6 2418.75   324.1 2419.14
   329.3 2420.88   349.7  2437.2     366 2447.43   374.1 2449.44   388.6 2455.75
   419.2  2466.7   454.6 2484.13     470 2490.34   480.5 2495.97   513.4 2511.32
#Mann= 3 ,-1,0
       0      .1       0   293.6    .045       0   324.1      .1       0
Bank Sta=293.6,324.1
XS Rating Curve= 0 ,0
Exp/Cntr(USF)=0,0
Exp/Cntr=0.3,0.1

Type RM Length L Ch R = 1 ,4192    ,70.6,71.1,72.1
XS GIS Cut Line= 3
2334612.10060885701757.0408382422334249.88583687701644.703851307
2334119.54612767701642.543524635
#Sta/Elev= 30
       0 2529.18      25 2522.99    33.4 2522.59    54.4 2516.98   140.5 2488.95
   169.2 2474.08   175.8 2471.43   184.2 2465.63   191.6 2461.72   230.3 2447.81
   238.6 2443.26     247 2443.06   252.4 2441.53   263.8 2435.26   276.3 2426.53
   288.9 2415.77   296.6 2411.82   301.5 2410.63   310.1 2410.21   316.3 2409.87
   322.7 2410.16   330.8 2413.97   347.5 2428.15   351.7 2429.71   360.1 2430.83
   368.5 2435.73   392.3    2447     481 2501.91   494.6 2508.57   509.6 2517.31
#Mann= 3 ,-1,0
       0      .1       0   310.1    .045       0   322.7      .1       0
Bank Sta=310.1,322.7
XS Rating Curve= 0 ,0
Exp/Cntr(USF)=0,0
Exp/Cntr=0.3,0.1

Type RM Length L Ch R = 1 ,4120    ,98.5,99.1,98.6
XS GIS Cut Line= 3
2334604.61147638701718.2269690392334308.35867879701584.430737164
 2334135.8205886701571.180733577
#Sta/Elev= 30
       0 2521.76    13.2 2519.09    53.1 2505.29      97 2493.64   132.1 2481.28
   158.3 2466.91   167.3 2464.98     176 2460.08   206.8 2449.21   218.8 2442.38
   228.7 2441.62   233.1 2439.69   245.5 2428.67   255.2 2411.03   258.1 2410.21
   272.6 2412.54   288.4 2406.13   294.1 2405.75   298.9 2406.22   307.7 2408.84
   329.3 2411.47   337.3 2415.14   353.3 2425.37   361.4 2426.89   373.4 2436.72
   385.4 2443.12   397.5 2453.57   413.5 2464.32   429.6 2471.91   498.1 2514.01
#Mann= 3 ,-1,0
       0      .1       0   288.4    .045       0   298.9      .1       0
Bank Sta=288.4,298.9
XS Rating Curve= 0 ,0
Exp/Cntr(USF)=0,0
Exp/Cntr=0.3,0.1

Type RM Length L Ch R = 1 ,4021    ,50,50.4,50.6
XS GIS Cut Line= 4
2334622.07360886701666.5871413232334395.23930832701520.765090971
2334341.44717419701493.5449749062334194.32892783701479.934916873
#Sta/Elev= 30
       0 2514.99    30.8  2505.5    40.3 2501.56    49.8 2499.94    83.1 2490.81
   121.1 2478.84   135.8 2472.39   155.8 2460.72   163.9 2458.96   180.1 2450.32
   193.4 2445.32   202.1 2439.31   228.2 2433.65   249.5 2421.85   268.6 2406.38
   274.6 2402.93   277.6 2401.97   286.6 2402.52   298.4 2400.04   304.4 2399.16
     309 2400.04   322.4 2404.01   339.3 2414.56   363.4 2425.49   371.4 2426.24
   375.4 2427.84   383.4 2433.16   419.5 2448.48   431.7 2455.59   477.7 2478.42
#Mann= 3 ,-1,0
       0      .1       0   298.4    .045       0     309      .1       0
Bank Sta=298.4,309
XS Rating Curve= 0 ,0
Exp/Cntr(USF)=0,0
Exp/Cntr=0.3,0.1

Type RM Length L Ch R = 1 ,3971    ,83.3,82.8,81.8
XS GIS Cut Line= 3
2334656.17127296701627.9973250452334372.44837006701451.570646845
2334204.66299855701419.165746768
#Sta/Elev= 30
       0 2513.63    37.7 2501.33    51.4 2498.37    65.9 2492.72    83.4 2488.65
   131.9 2471.54   174.3 2453.32   183.7 2451.01   193.1 2445.01   202.4 2441.25
   214.1 2439.55   225.7 2430.71   240.2 2428.26   263.4 2407.62   282.6 2393.99
     292 2390.75   308.3 2389.99   312.8 2389.63  317.292390.003   334.4 2398.55
   346.6 2402.67   362.9 2413.38   375.1 2419.47   391.4 2425.06   403.6    2426
     424 2435.67   466.1 2451.39   485.1 2461.91   493.3 2463.41     505 2470.07
#Mann= 3 ,-1,0
       0      .1       0   308.3    .045       0  317.29      .1       0
Bank Sta=308.3,317.29
XS Rating Curve= 0 ,0
Exp/Cntr(USF)=0,0
Exp/Cntr=0.3,0.1

Type RM Length L Ch R = 1 ,3888    ,105.9,105.5,104.5
XS GIS Cut Line= 4
2334681.23106235701584.9348133862334527.12775976 701458.91575753
2334434.23371287  701399.86682852334247.00540131701336.497246126
#Sta/Elev= 30
       0 2509.16      29  2498.1    37.5 2496.66      53 2490.83    91.5 2478.94
   144.9 2457.85   171.9  2448.8   182.5 2443.39   193.9 2441.78     212 2431.56
   221.5 2423.71   226.3 2422.05   235.7  2421.3   239.6 2419.03     250 2411.17
   268.9  2394.2   274.9 2387.44   278.4 2385.32   287.9 2384.84   291.8 2385.25
   311.3 2390.46   319.2 2394.53   340.9 2403.06     362 2409.62   387.3 2420.62
   404.2 2422.71     417 2428.95   463.3  2442.4   486.4 2452.59   506.8 2459.86
#Mann= 3 ,-1,0
       0      .1       0   278.4    .045       0   291.8      .1       0
Bank Sta=278.4,291.8
XS Rating Curve= 0 ,0
Exp/Cntr(USF)=0,0
Exp/Cntr=0.3,0.1

Type RM Length L Ch R = 1 ,3783    ,91,92.7,94.2
XS GIS Cut Line= 3
2334722.83735381701513.083948524 2334562.4130954701352.339641719
2334318.29618148701221.999932519
#Sta/Elev= 30
       0 2498.28    15.1 2492.09    66.1 2478.58   103.6 2462.68   123.4    2456
   135.5 2454.56   169.4 2442.48     185 2434.52     202 2428.76   220.3 2418.99
     234 2407.83   238.7 2406.24   251.8 2405.21   263.6 2395.47   299.1 2380.64
     305 2379.85  309.692380.633   320.3 2383.56   338.5 2392.94   352.3 2402.24
   369.7 2408.01   375.9  2411.7   383.8    2413   397.4  2412.7     411 2418.31
   447.3 2423.54   465.4 2428.53   474.5 2428.13   483.6 2434.76   503.8 2445.17
#Mann= 3 ,-1,0
       0      .1       0   299.1    .045       0  309.69      .1       0
Bank Sta=299.1,309.69
XS Rating Curve= 0 ,0
Exp/Cntr(USF)=0,0
Exp/Cntr=0.3,0.1

Type RM Length L Ch R = 1 ,3690    ,154.3,153.2,149.3
XS GIS Cut Line= 5
2334732.21089837701497.4150002482334705.80690571701419.803264261
2334594.59008816701286.1830590032334537.40363374701228.152090933
 2334353.7536703701144.561643849
#Sta/Elev= 30
       0  2494.4    12.8 2490.38    72.1  2476.1    90.6 2470.23     101 2469.16
   116.6  2464.9   159.6 2449.44   178.3 2438.48   222.1 2418.07   236.3 2408.36
   246.9 2397.97   251.9 2395.07     265 2392.98   283.7 2381.94   296.5 2377.33
   306.12376.124   310.6 2375.73   317.32376.124     329 2379.44   347.4  2392.2
   361.6 2397.74   379.7 2401.71   391.8 2405.84   403.9 2406.97   413.4  2411.7
   474.9 2430.85   488.5  2436.2   500.5  2438.1   523.2 2444.67   539.1 2447.65
#Mann= 3 ,-1,0
       0      .1       0   306.1    .045       0   317.3      .1       0
Bank Sta=306.1,317.3
XS Rating Curve= 0 ,0
Exp/Cntr(USF)=0,0
Exp/Cntr=0.3,0.1

Type RM Length L Ch R = 1 ,3537    ,104.9,110.5,121.1
XS GIS Cut Line= 3
2334746.84098349701455.4752372752334650.02634376701127.425631552
2334427.59270866701041.012564679
#Sta/Elev= 30
       0 2484.64    39.4 2473.85    73.3 2467.92      90 2462.51   102.5 2459.93
   144.2 2448.63   194.2  2432.6   202.6 2431.23   213.3 2427.76   256.8 2407.88
   269.3 2400.71   273.5 2397.62   287.4 2383.09   294.3 2378.31   315.2 2373.99
   345.2 2369.57  359.522365.926   361.2 2365.66  371.152365.904   378.4 2367.83
   395.5 2385.19   399.8 2388.87   404.1 2390.91   414.5 2394.13   425.6 2394.31
   428.6 2395.08   481.2 2412.63   498.5 2419.97   528.5 2431.15   580.7 2447.03
#Mann= 3 ,-1,0
       0      .1       0  359.52    .045       0  371.15      .1       0
Bank Sta=359.52,371.15
XS Rating Curve= 0 ,0
Exp/Cntr(USF)=0,0
Exp/Cntr=0.3,0.1

Type RM Length L Ch R = 1 ,3426    ,134.9,130.5,120.8
XS GIS Cut Line= 5
2334756.44243537701433.0718495672334710.36349263701090.974919439
2334718.49358576701056.0807021162334705.11035372701016.935313195
2334504.40432366700920.994416244
#Sta/Elev= 30
       0 2479.57      16 2475.71    28.1 2470.19    56.4 2465.45    72.5  2460.5
     121 2443.78   157.3 2429.52   169.4 2427.35   193.6 2418.33   214.1 2407.28
     230 2403.63   242.1 2394.82   250.1 2386.55   270.3 2375.79   282.4 2367.21
   301.7 2363.33   322.8 2362.36   334.5 2363.64   360.42360.102   367.6 2359.67
  371.74  2360.1   388.4 2364.01   409.4 2376.33   413.7 2377.54   445.6 2379.36
   470.9 2382.88   497.9  2388.3   512.1 2392.52   551.7 2406.39   644.8    2446
#Mann= 3 ,-1,0
       0      .1       0   360.4    .045       0  371.74      .1       0
#XS Ineff= 2 , 0
          332.52  2367.4
Permanent Ineff=
       F       F
Bank Sta=360.4,371.74
XS Rating Curve= 0 ,0
Exp/Cntr(USF)=0,0
Exp/Cntr=0.3,0.1

Type RM Length L Ch R = 1 ,3296    ,97.7,96.3,94.3
XS GIS Cut Line= 3
2335037.10996283701043.4731544872334872.28503898701045.873517456
 2334517.8314406 700908.25270725
#Sta/Elev= 30
       0 2467.75    16.9 2459.94    32.9 2450.63      46 2444.42    68.9 2430.55
   100.9 2413.97     145 2397.58     153 2393.85   169.3 2381.88   199.3 2354.03
   203.6 2351.98  213.05 2350.38   216.5 2349.66   221.62350.382   233.5 2351.11
   242.2 2354.13   267.9 2365.89   280.8 2366.58     286 2368.59   298.4 2370.76
   306.6 2374.86   310.4 2375.81     328 2375.23   340.9 2376.17   366.4 2379.03
     401 2385.88   459.1 2406.33   499.7 2423.65   508.2 2428.25   545.1  2444.3
#Mann= 3 ,-1,0
       0      .1       0  213.05    .045       0   221.6      .1       0
Bank Sta=213.05,221.6
XS Rating Curve= 0 ,0
Exp/Cntr(USF)=0,0
Exp/Cntr=0.3,0.1

Type RM Length L Ch R = 1 ,3200    ,83.6,84.7,86
XS GIS Cut Line= 4
2335058.88816943700989.0047003582334880.46118875700939.397199004
2334793.24800089700931.3959891092334569.21412381700839.382075309
#Sta/Elev= 30
       0 2471.24       7 2466.43    21.6 2461.13    73.4  2429.2    94.2 2417.46
   102.5 2413.99   151.5  2380.2   168.9 2363.61   197.5 2345.12   205.2 2342.52
   209.6 2341.97   217.6 2342.46   229.7 2347.31   245.7 2359.49   249.8 2360.67
   257.8 2360.43   261.8 2362.34   269.8 2368.75   278.3 2371.46   317.2 2371.22
   342.7 2372.48   352.3 2373.37   377.7 2378.85     404 2390.35   416.3 2393.45
   429.6 2399.58   436.5 2401.46   456.1 2413.16   468.4 2416.83     515 2436.67
#Mann= 3 ,-1,0
       0      .1       0   205.2    .045       0   217.6      .1       0
Bank Sta=205.2,217.6
XS Rating Curve= 0 ,0
Exp/Cntr(USF)=0,0
Exp/Cntr=0.3,0.1

Type RM Length L Ch R = 1 ,3115    ,103.5,103,102.5
XS GIS Cut Line= 3
2335078.09107318700912.9932063492334825.25284047700840.982317288
 2334600.4188424700764.170702289
#Sta/Elev= 30
       0  2466.6    39.4 2444.48    56.1 2433.05    68.5 2426.32      81 2417.72
    93.5 2411.51   122.6 2392.97   151.7    2373   185.9 2344.79   189.1 2342.88
  202.592339.953   205.8 2339.62   211.8  2339.9   226.6 2340.04   243.2 2349.02
   255.7 2350.98   268.3 2363.02   280.9 2368.34   297.8 2370.23   310.8 2366.25
   327.4 2365.92   361.3 2373.53   378.2  2379.4   395.1 2388.34   437.3 2401.21
   441.6 2403.45     450 2410.68   458.5 2412.86   479.6 2422.29   500.5  2426.7
#Mann= 3 ,-1,0
       0      .1       0  202.59    .045       0   211.8      .1       0
Bank Sta=202.59,211.8
XS Rating Curve= 0 ,0
Exp/Cntr(USF)=0,0
Exp/Cntr=0.3,0.1

Type RM Length L Ch R = 1 ,3012    ,145,142.6,138.5
XS GIS Cut Line= 3
2335112.49627573700837.7818333292334923.66772219700759.369976352
2334620.42186714700712.162837968
#Sta/Elev= 30
       0 2462.62       9 2456.47      22 2452.07      48 2435.16    65.3 2426.33
    82.6 2415.33    91.3 2411.89   126.2 2389.95   143.3 2380.94   177.9 2359.76
   199.7 2347.56   224.2 2336.42     234 2333.76   240.4 2333.27  245.532333.804
   251.5 2335.93   256.6 2339.42     269 2341.78   272.8 2344.38   284.9 2357.38
     289 2360.77     293 2362.57   341.6  2367.8   365.9 2373.99   394.2 2383.26
   434.7 2400.43   454.9 2404.79   467.1 2412.12   479.2 2417.53   511.4  2426.9
#Mann= 3 ,-1,0
       0      .1       0     234    .045       0  245.53      .1       0
Bank Sta=234,245.53
XS Rating Curve= 0 ,0
Exp/Cntr(USF)=0,0
Exp/Cntr=0.3,0.1

Type RM Length L Ch R = 1 ,2869    ,129.1,133.4,136.4
XS GIS Cut Line= 4
2335157.30305114700696.9605391662334946.87123089700608.147109324
2334846.85610719700640.1519489062334647.62598079700613.747956251
#Sta/Elev= 30
       0  2437.5      19 2428.16    28.2  2425.7      36 2420.83      49 2417.82
    58.7 2412.49    79.4 2403.68      92 2396.05   114.1 2385.08   180.8 2355.01
     190 2349.93   200.9 2346.56   218.3 2338.06   235.4 2333.86     248 2327.92
  250.242327.856     260 2327.62  263.812327.885     269 2328.99   281.6 2327.79
     290 2330.04     332 2354.84   352.3 2357.83     361 2360.33   408.8 2377.73
   434.6 2392.05   473.3 2410.74   484.5 2413.55   521.7 2428.31   534.4 2431.55
#Mann= 3 ,-1,0
       0      .1       0  250.24    .045       0  263.81      .1       0
Bank Sta=250.24,263.81
XS Rating Curve= 0 ,0
Exp/Cntr(USF)=0,0
Exp/Cntr=0.3,0.1

Type RM Length L Ch R = 1 ,2736    ,118.7,120.7,122.1
XS GIS Cut Line= 2
2335182.90692281700608.1471093242334698.83372412700440.921822504
#Sta/Elev= 30
       0 2427.43    19.8 2419.31    32.5 2416.32    61.1 2405.64    70.6 2402.86
   138.3 2366.97   172.2 2352.54   193.2 2346.85   237.2 2337.47     253 2335.45
   256.8 2334.21   265.3 2329.21   268.7 2328.27   281.3 2328.14   303.4 2324.58
  323.822319.071   327.6  2318.7   335.8 2319.05   341.4 2320.62   349.9 2325.58
   358.4 2332.37   375.3 2343.84   396.5 2361.91   426.3 2380.63     443  2390.2
   455.7 2394.88   465.1 2401.04   476.9  2405.6   481.1  2408.3   512.1 2423.13
#Mann= 3 ,-1,0
       0      .1       0  323.82    .045       0   335.8      .1       0
Bank Sta=323.82,335.8
XS Rating Curve= 0 ,0
Exp/Cntr(USF)=0,0
Exp/Cntr=0.3,0.1

Type RM Length L Ch R = 1 ,2615    ,98.4,97.8,96.3
XS GIS Cut Line= 3
2335192.50837468700565.7406968772334896.46360854700376.912143339
2334724.43759579700332.105367923
#Sta/Elev= 30
       0 2420.98    12.2 2416.07    52.8 2406.57    71.6  2400.7    97.7 2388.25
   119.4 2375.78   133.2 2370.61     160 2355.58   194.7 2339.17   223.4  2333.3
   246.9 2331.37   256.6 2325.09   270.8 2321.87   284.5 2313.52   288.52311.983
   293.2 2311.49   297.22311.975   327.8 2312.41   345.4  2319.6   380.7 2344.19
   388.6 2350.58   397.1 2355.13   413.4 2366.43   430.2 2372.56   450.6 2384.69
   471.3 2394.26   482.3 2401.02   500.2 2409.17   511.8 2415.74   528.9 2421.38
#Mann= 3 ,-1,0
       0      .1       0   288.5    .045       0   297.2      .1       0
Bank Sta=288.5,297.2
XS Rating Curve= 0 ,0
Exp/Cntr(USF)=0,0
Exp/Cntr=0.3,0.1

Type RM Length L Ch R = 1 ,2517    ,169.4,172.6,165.9
XS GIS Cut Line= 2
2335236.51502911700396.9151680782334758.04267735700249.692905998
#Sta/Elev= 30
       0 2384.87    17.1 2379.89      38 2372.46    67.3 2364.58   109.7 2350.49
   138.5 2343.94   171.9 2332.31   201.7 2324.56   205.4 2323.27   213.8 2318.68
   220.9 2316.47   230.5 2312.36   234.7 2311.52   243.1 2312.13   252.9 2308.82
   266.9 2306.37   272.4 2305.61  281.012306.351   305.9 2320.69     331 2339.92
   347.7 2350.34   363.6  2358.1   377.7 2363.53   389.6 2366.86   397.9 2371.25
   414.7 2377.74   439.8 2389.51   448.3 2392.18   456.5 2395.93   500.6  2410.8
#Mann= 3 ,-1,0
       0      .1       0   266.9    .045       0  281.01      .1       0
Bank Sta=266.9,281.01
XS Rating Curve= 0 ,0
Exp/Cntr(USF)=0,0
Exp/Cntr=0.3,0.1

Type RM Length L Ch R = 1 ,2345    ,99.2,99.8,101.5
XS GIS Cut Line= 3
2335292.52349838700272.0962937062335101.29458187700195.284678707
2334809.25042068700161.679597146
#Sta/Elev= 30
       0 2407.25    34.9 2392.19    47.8 2383.32      65 2375.76    73.7 2372.49
    86.6  2369.9    91.7 2367.97   104.4 2360.46   116.8 2355.65     134 2345.14
   142.6 2341.28   172.8 2324.82   197.1 2310.26   215.3  2300.5  220.69 2299.28
   231.4 2298.43   235.4 2299.28   243.4 2301.32   251.5 2300.52   263.2 2303.43
   303.8 2326.27     332 2337.41   346.2 2341.94   364.2 2350.25   396.8 2359.59
   408.5 2364.59   432.7  2371.7   448.8  2373.4   465.4  2377.7   500.1 2391.28
#Mann= 3 ,-1,0
       0      .1       0  220.69    .045       0   235.4      .1       0
#XS Ineff= 2 , 0
                           243.7         2305.48
Permanent Ineff=
       F       F
Bank Sta=220.69,235.4
XS Rating Curve= 0 ,0
Exp/Cntr(USF)=0,0
Exp/Cntr=0.3,0.1

Type RM Length L Ch R = 1 ,2245    ,95.7,94.7,93.6
XS GIS Cut Line= 4
2335316.09838931700179.0528328282335127.26983577 700102.24121783
 2335029.4774736700074.7556462952334852.52005127700057.486058302
#Sta/Elev= 30
       0 2402.46    16.7 2393.67      69  2368.9      82 2363.94    94.9 2355.64
   120.8 2341.97   139.5 2330.59   181.3 2308.88   211.2 2297.07   220.2 2294.14
   223.7 2293.81     2332294.069   236.2 2293.91   248.6 2297.66   256.9  2298.3
   265.6 2297.86   273.5 2299.08   285.1 2304.46   294.3 2310.08   306.7 2316.29
   314.8 2319.01     359 2337.48   375.1  2346.2   391.1 2353.16   419.3 2367.74
   447.6  2379.3   467.5 2386.45   475.5 2391.41   479.6 2392.48   483.2 2392.32
#Mann= 3 ,-1,0
       0      .1       0   220.2    .045       0     233      .1       0
Bank Sta=220.2,233
XS Rating Curve= 0 ,0
Exp/Cntr(USF)=0,0
Exp/Cntr=0.3,0.1

Type RM Length L Ch R = 1 ,2150    ,112.6,112.9,111.1
XS GIS Cut Line= 4
2335353.04555853700082.5483094722335172.50534994700008.056367149
2335007.68042609699995.2544313162334828.73685834700015.779364996
#Sta/Elev= 30
       0 2410.61     9.6 2408.07    20.1 2401.89    35.4 2395.75    57.2    2382
    87.5  2366.9   108.9 2354.51   152.4 2327.24   170.2 2317.49   178.4 2311.56
   191.3 2299.27   199.6 2293.73   219.7 2290.65   240.4 2290.07   243.8 2289.61
  249.05 2290.04   267.9 2297.81   279.9  2299.2   283.9 2301.42   295.9 2310.83
   299.9 2312.76     304 2313.69   332.3 2312.84   352.1 2316.47   376.4 2327.58
   387.2 2334.57   436.6 2362.62   484.9 2381.58   509.1 2390.19   540.7 2399.86
#Mann= 3 ,-1,0
       0      .1       0   240.4    .045       0  249.05      .1       0
Bank Sta=240.4,249.05
XS Rating Curve= 0 ,0
Exp/Cntr(USF)=0,0
Exp/Cntr=0.3,0.1

Type RM Length L Ch R = 1 ,2037    ,91.2,89.2,88
XS GIS Cut Line= 4
2335369.17181149699947.784243243 2335186.6432186699901.788584051
2335006.84477145 699889.483457692334852.95750461699942.834790815
#Sta/Elev= 30
       0 2403.43    16.1 2396.93    29.9 2392.66    50.5 2380.34    62.9 2374.07
   125.3 2334.18   174.3 2300.57   190.7 2288.16   194.7 2286.05  207.722283.334
   210.8 2282.87   220.4 2283.35   230.8 2285.53   234.8 2287.78   238.8 2291.07
   254.8 2300.15   262.9 2300.46   266.9  2301.5   274.9 2306.02   278.9 2307.45
     299 2307.16     327 2308.41   339.1 2310.88   363.1 2313.45   379.8 2317.75
   392.3 2322.78   422.1 2338.36   467.8 2359.52   502.5 2372.15   531.3 2381.14
#Mann= 3 ,-1,0
       0      .1       0  207.72    .045       0   220.4      .1       0
Bank Sta=207.72,220.4
XS Rating Curve= 0 ,0
Exp/Cntr(USF)=0,0
Exp/Cntr=0.3,0.1

Type RM Length L Ch R = 1 ,1948    ,131.6,129.8,129.2
XS GIS Cut Line= 4
2335414.19928429699847.6841386972335182.29651747699809.625408801
2335005.27041827699837.0042599352334843.73622223699899.085511308
#Sta/Elev= 30
       0 2403.23    72.2 2380.51    94.5 2371.08     148 2344.54   188.4  2317.9
   200.7 2306.78     225 2290.41   233.1 2283.15   237.2 2277.88241.16322275.382
   245.2  2274.8255.12982275.402   265.5 2277.11   273.6 2279.77   289.8 2287.61
   301.9 2295.89     306 2297.08   314.1  2297.2   327.6 2301.55   338.3  2303.7
   378.8 2307.52   419.6  2313.4   449.2 2319.89   466.7 2327.63   488.2  2335.4
   498.7 2337.99   509.6 2343.23   518.2 2345.58     561 2362.47   587.2 2371.59
#Mann= 3 ,-1,0
       0      .1       0241.1632    .045       0255.1298      .1       0
Bank Sta=241.1632,255.1298
XS Rating Curve= 0 ,0
Exp/Cntr(USF)=0,0
Exp/Cntr=0.3,0.1

Type RM Length L Ch R = 1 ,1818    ,148.3,149.8,150.9
XS GIS Cut Line= 3
2335413.34907966699729.9489150622335159.90489757699678.778884931
2334822.99586517699785.846284532
#Sta/Elev= 30
       0 2394.98    21.6 2387.11    33.8 2384.58    46.1 2378.78    62.8 2373.73
    74.7 2366.25    82.8    2364   131.8 2342.62   148.1 2334.41     193 2307.97
   221.6  2296.7   258.3 2279.69   266.6 2269.99   270.9 2266.74   282.5 2266.24
   303.7 2266.73   311.2  2269.9   321.2 2276.38   329.6 2279.28   350.6 2283.96
   362.2 2284.03   396.8 2288.66   413.6 2294.44   435.4 2305.74   486.4 2319.53
   531.1  2334.1   543.7 2336.49   564.7  2344.2   585.7 2348.32   612.1 2357.96
#Mann= 3 ,-1,0
       0      .1       0   270.9    .045       0   303.7      .1       0
Bank Sta=270.9,303.7
XS Rating Curve= 0 ,0
Exp/Cntr(USF)=0,0
Exp/Cntr=0.3,0.1

Type RM Length L Ch R = 1 ,1669    ,93.7,93.6,94.1
XS GIS Cut Line= 4
2335410.18827776 699637.397940462335233.76159956 699554.58541804
2335060.21535692699549.5446558052334818.97887857699640.278376022
#Sta/Elev= 30
       0 2379.24    50.8 2364.42    86.2 2351.47   195.1 2308.43   208.5 2302.27
   256.5 2286.48   272.5 2275.45   280.5 2272.26   300.5 2266.92   320.5 2264.26
   337.8 2259.92   340.5 2259.52   345.6 2259.96   352.5 2261.84   360.6 2266.66
   380.7  2274.2   394.2 2273.16   398.5 2274.92     407 2281.78   411.3 2283.51
   424.1  2285.2   445.5 2282.86     454 2283.75   481.1 2292.31   522.4 2301.59
   551.5 2310.98     578 2325.14   594.7 2340.03   617.4 2353.68   626.3 2357.93
#Mann= 3 ,-1,0
       0      .1       0   337.8    .045       0   345.6      .1       0
Bank Sta=337.8,345.6
XS Rating Curve= 0 ,0
Exp/Cntr(USF)=0,0
Exp/Cntr=0.3,0.1

Type RM Length L Ch R = 1 ,1575    ,88.3,88.1,88.3
XS GIS Cut Line= 2
2335418.82958445699478.2538756352334830.50062082699440.808213323
#Sta/Elev= 30
       0 2364.31    67.6  2340.4    87.3 2334.43    94.8 2331.14   102.9 2326.02
   114.9 2323.43   126.9 2319.04   138.9 2313.65     163 2305.16     175 2299.05
   203.1 2293.73   239.1 2279.27   247.2 2273.58     256 2269.83   267.2 2266.61
   283.2 2263.83   323.3 2259.44  334.172256.248   339.3 2255.86   343.3 2256.24
   363.4 2258.61   379.4 2265.84   395.5    2268   407.5 2274.53   483.6 2302.96
   502.5 2311.69   515.4 2316.38   523.7  2320.9   547.8 2328.62   589.5 2348.11
#Mann= 3 ,-1,0
       0      .1       0  334.17    .045       0   343.3      .1       0
Bank Sta=334.17,343.3
XS Rating Curve= 0 ,0
Exp/Cntr(USF)=0,0
Exp/Cntr=0.3,0.1

Type RM Length L Ch R = 1 ,1487    ,140.5,139.1,137.4
XS GIS Cut Line= 2
2335421.71002001699403.3625510122334842.74247196699345.033730872
#Sta/Elev= 30
       0 2366.18    33.7 2352.68    50.9 2348.25    69.9  2340.4    87.4 2334.56
   106.1 2326.23   134.2 2316.24   173.6 2299.51   186.5 2295.21   202.6 2286.44
   222.5 2269.45   236.2 2262.64   242.8 2261.02     295 2258.93   317.5 2251.89
   323.2 2251.33   328.4 2251.87   343.3 2254.03   359.3 2254.74   379.4 2261.47
   415.6 2262.84   428.5 2267.84   443.8  2276.5   452.6  2283.4   489.2 2306.73
   514.7 2325.14   528.2 2336.02   536.2 2340.48   552.3 2353.49   581.9 2372.74
#Mann= 3 ,-1,0
       0      .1       0   317.5    .045       0   328.4      .1       0
Bank Sta=317.5,328.4
XS Rating Curve= 0 ,0
Exp/Cntr(USF)=0,0
Exp/Cntr=0.3,0.1

Type RM Length L Ch R = 1 ,1348    ,131.2,134.4,136.2
XS GIS Cut Line= 4
2335431.03154955699250.465151803 2335161.7507105 699224.05543725
2335068.13655472699240.6179417342334845.97156867699223.126496061
#Sta/Elev= 30
       0 2374.25      23 2368.15    95.3 2336.68   127.5 2318.15   155.6 2300.17
   187.8 2283.57   199.8 2275.11   211.9 2265.04   227.9 2256.26     244 2252.24
   292.5 2247.81   308.7 2248.54   320.9 2247.53     329  2245.7   337.2 2245.33
   341.9 2245.69   353.4 2248.31   365.6 2255.24   393.7 2255.73   409.8 2257.73
   433.8 2264.92   453.9 2273.26   469.9  2283.1     482 2289.01     490 2294.31
   518.1 2317.14   534.1 2328.59   570.2  2359.3   582.3  2368.6   588.5 2372.27
#Mann= 3 ,-1,0
       0      .1       0     329    .045       0   341.9      .1       0
#XS Ineff= 2 , 0
          308.45  2258.1
Permanent Ineff=
       F       F
Bank Sta=329,341.9
XS Rating Curve= 0 ,0
Exp/Cntr(USF)=0,0
Exp/Cntr=0.3,0.1

Type RM Length L Ch R = 1 ,1213    ,89.7,88.5,88.4
XS GIS Cut Line= 4
2335424.59045557699140.5228059392335188.39473945699121.799974783
2335033.57132797699090.1151835962334858.58486755699126.120628126
#Sta/Elev= 30
       0 2370.77     9.9 2369.81    28.5 2365.07    48.1 2354.54    88.7 2336.62
   128.8 2314.61   136.3 2308.97   144.9 2300.87   152.9 2295.95     173 2286.76
     201    2276   213.1  2269.7   237.6 2249.84   253.5 2245.05   269.8 2244.77
   286.2 2243.31   302.5 2239.09   310.7 2238.65  316.172239.046   331.1 2245.15
   380.1 2245.97   392.3 2248.73   408.6 2257.53   446.2  2273.2     480 2289.46
   494.4 2294.86   517.3 2306.03   536.8 2317.59   559.7 2333.73   573.6 2342.27
#Mann= 3 ,-1,0
       0      .1       0   302.5    .045       0  316.17      .1       0
Bank Sta=302.5,316.17
XS Rating Curve= 0 ,0
Exp/Cntr(USF)=0,0
Exp/Cntr=0.3,0.1

Type RM Length L Ch R = 1 ,1125    ,84.6,85,85.4
XS GIS Cut Line= 3
2335410.90838665699065.6314813152335014.12838792699001.541790051
2334865.78595646699039.707561253
#Sta/Elev= 30
       0 2361.42    10.9 2358.97      23 2358.38    27.1 2356.08    39.2 2346.15
    47.3 2341.42    72.5 2329.76    87.9 2323.86   144.6 2292.77   197.3  2271.8
   221.6 2256.77   245.9 2243.61   262.1 2238.93   274.2 2238.62   290.4 2235.25
   298.6 2235.05  299.742235.305   310.7 2240.67   322.9 2240.65     331 2242.62
   351.2 2241.16   367.4 2242.73   383.6 2245.61   395.8 2249.25   408.1  2250.6
   465.6 2280.19   494.8  2290.8   515.5 2294.28   531.3 2302.44   555.1 2312.01
#Mann= 3 ,-1,0
       0      .1       0   290.4    .045       0  299.74      .1       0
Bank Sta=290.4,299.74
XS Rating Curve= 0 ,0
Exp/Cntr(USF)=0,0
Exp/Cntr=0.3,0.1

Type RM Length L Ch R = 1 ,1040    ,102.7,100.1,97.2
XS GIS Cut Line= 3
2335400.82686218698997.2211367072335055.17459469698916.568940959
 2334847.0631253698975.617869989
#Sta/Elev= 30
       0 2352.22    29.4 2342.49    53.9 2339.11    58.2 2337.37    70.5 2329.21
   115.7 2308.46   148.5 2289.71     183 2274.79   222.5 2254.39   230.4  2247.7
   234.8 2241.08   238.9  2236.6   247.1 2234.46   263.5 2235.09   270.3  2232.7
   275.9 2232.18  280.932232.653   288.2 2235.83     297 2236.34   308.7 2239.64
   337.5 2239.16   374.7 2241.45   416.2 2251.86   424.6 2255.33   437.1 2256.94
   449.5 2266.07   458.3 2269.13   480.9 2282.78   495.3 2290.11   571.3 2311.34
#Mann= 3 ,-1,0
       0      .1       0   270.3    .045       0  280.93      .1       0
Bank Sta=270.3,280.93
XS Rating Curve= 0 ,0
Exp/Cntr(USF)=0,0
Exp/Cntr=0.3,0.1

Type RM Length L Ch R = 1 ,940     ,165.2,161.2,161
XS GIS Cut Line= 3
2335408.74805998698901.4466542562335180.47354166698824.395002961
2334844.90279863698907.927634272
#Sta/Elev= 30
       0 2350.12    30.2 2340.27    76.6 2320.44   101.9 2314.22   125.9 2301.55
   190.6 2272.42     199 2267.38   215.9 2254.49   228.6 2240.57   241.2 2238.42
   249.5  2233.4   253.6 2232.41   270.1 2232.46   282.5 2230.96   290.7 2230.67
   294.8 2230.99   303.1 2234.68   307.2 2235.23   331.9 2233.26   356.7 2236.86
   389.6 2238.58   403.5 2240.53   426.6 2248.74     463 2257.22   476.2 2263.62
   488.6 2265.11     505 2277.36     538 2291.49   554.5 2295.41   586.7 2300.41
#Mann= 3 ,-1,0
       0      .1       0   282.5    .045       0   294.8      .1       0
#XS Ineff= 2 , 0
           269.6 2238.92  307.28          2239.7
Permanent Ineff=
       F       F
Bank Sta=282.5,294.8
XS Rating Curve= 0 ,0
Exp/Cntr(USF)=0,0
Exp/Cntr=0.3,0.1

Type RM Length L Ch R = 1 ,779     ,114,116.7,122.1
XS GIS Cut Line= 4
2335405.86762442 698788.389558432335122.86483041698668.131373698
2334986.04414119698765.3460739312334826.17996747698842.397725226
#Sta/Elev= 30
       0 2333.09      41 2320.79    58.3 2313.35    71.4 2311.07    93.1 2303.85
   110.5 2294.66   127.9  2288.7   149.6 2285.04   197.4 2264.42   214.8  2251.9
   249.6 2247.75   271.3 2235.33   288.7 2234.45   320.6 2228.95   367.5 2226.18
   379.5 2227.87   399.1 2227.38   413.4 2224.59   433.6 2224.02   447.4 2220.81
   454.3 2220.22   461.2 2220.73     475 2234.25   482.6 2238.78   542.5  2260.3
   561.8 2268.12   575.5 2276.29   590.5 2278.77   622.4 2291.08   652.8  2297.8
#Mann= 3 ,-1,0
       0      .1       0   447.4    .045       0   461.2      .1       0
Bank Sta=447.4,461.2
XS Rating Curve= 0 ,0
Exp/Cntr(USF)=0,0
Exp/Cntr=0.3,0.1

Type RM Length L Ch R = 1 ,662     ,101.3,101.5,101.5
XS GIS Cut Line= 3
2335400.82686218698745.1830249942335165.35125495698642.207453636
2334765.69082066698642.927562527
#Sta/Elev= 30
       0 2325.12    31.3 2317.32    55.2 2308.92   109.9 2293.72     123 2288.57
   136.1 2279.61   153.5 2277.53   166.6 2273.49   173.6 2268.97   192.8 2260.21
   205.9 2250.77   228.3 2247.85   266.2 2236.83   279.3 2234.94   294.2 2230.35
     337 2226.39   418.2 2222.56   442.2  2215.6   450.2 2214.72   455.6  2215.6
   482.2 2228.02   507.7  2246.6   514.2 2252.54   530.2 2275.08   534.2 2279.21
   540.6 2283.05   558.2 2290.93   582.2 2293.28   590.2 2295.77   656.7 2326.06
#Mann= 3 ,-1,0
       0      .1       0   442.2    .045       0   455.6      .1       0
Bank Sta=442.2,455.6
XS Rating Curve= 0 ,0
Exp/Cntr(USF)=0,0
Exp/Cntr=0.3,0.1

Type RM Length L Ch R = 1 ,560     ,87.5,90.7,92.3
XS GIS Cut Line= 3
2335421.71002001698698.3759471042335047.25339689698542.112317841
2334766.41092955698538.511773388
#Sta/Elev= 30
       0 2329.02     107 2299.83   127.4 2289.97   148.9 2283.74     162 2272.75
   192.4 2266.66     227 2247.62   235.7 2246.17   248.7 2240.79   271.2  2236.7
     311  2233.2   387.4 2232.22   404.8 2227.49   412.8 2221.31   416.8 2220.12
   456.6 2219.07   464.7 2217.57  472.362213.893   476.8 2213.13   486.32213.783
   492.8 2214.81   508.5 2222.11   524.3 2232.01   536.8  2244.4   544.8  2259.2
   552.8 2271.19   568.8 2283.68   596.8 2291.59   636.9 2297.86   686.6 2302.88
#Mann= 3 ,-1,0
       0      .1       0  472.36    .045       0   486.3      .1       0
Bank Sta=472.36,486.3
XS Rating Curve= 0 ,0
Exp/Cntr(USF)=0,0
Exp/Cntr=0.3,0.1

Type RM Length L Ch R = 1 ,470     ,119.5,121.2,123.3
XS GIS Cut Line= 3
2335429.17376066698678.0772054672334977.66548625698449.802687144
2334777.47521466698446.202142691
#Sta/Elev= 30
       0 2330.19    41.5 2321.94    90.8 2308.28   153.5 2281.49   162.5 2279.46
   175.9 2271.46   184.9 2269.33   198.3 2262.16   216.3 2258.27   239.6 2244.09
   261.1 2238.18   338.9 2228.98   377.6 2227.13   409.8 2216.48   467.3 2215.95
   480.7  2213.1   485.2 2210.75   495.6 2210.97   504.5 2210.32  508.45 2211.05
   543.4 2238.23   547.6 2246.41   551.4 2260.66   555.4 2267.84   583.4 2284.35
   603.4 2291.45   651.4 2302.97   671.5 2304.87   683.5 2308.45   706.2 2311.38
#Mann= 3 ,-1,0
       0      .1       0   495.6    .045       0  508.45      .1       0
Bank Sta=495.6,508.45
XS Rating Curve= 0 ,0
Exp/Cntr(USF)=0,0
Exp/Cntr=0.3,0.1

Type RM Length L Ch R = 1 ,348     ,96.5,93,89.1
XS GIS Cut Line= 4
2335419.77231651698586.2243965922335124.68083137 698413.08398439
2335016.27987764 698327.266562692334791.95012618698370.928057941
#Sta/Elev= 30
       0 2332.47     8.8 2328.93    27.4 2326.23      83 2302.04   112.7 2286.69
   137.8 2275.23     170 2264.12     185  2256.2   203.6 2244.36   208.2 2242.74
   226.8 2240.16   240.7 2233.27   259.2 2230.64   324.9 2228.44   333.7 2225.75
     353 2215.79   382.3  2213.3   398.9 2210.16   429.5 2209.36   439.2 2206.22
   449.9 2205.67  452.942206.204   464.9 2209.74   480.5 2222.75   488.7  2227.4
   500.9 2236.44   517.2 2250.94   533.5 2268.49   549.8 2278.91   708.9 2306.42
#Mann= 3 ,-1,0
       0      .1       0   439.2    .045       0  452.94      .1       0
Bank Sta=439.2,452.94
XS Rating Curve= 0 ,0
Exp/Cntr(USF)=0,0
Exp/Cntr=0.3,0.1

Type RM Length L Ch R = 1 ,255     ,93,93.1,93.1
XS GIS Cut Line= 6
2335481.83247428698560.2691884862335464.93938056698452.841962241
 2335246.0296581698319.2986690892335000.67770522698252.072234001
2334823.29953191698241.1305837222334743.89318821698335.789331968
#Sta/Elev= 30
       0 2330.52     7.2  2323.4    19.3  2319.5    39.1  2306.3    88.2 2278.48
   108.7 2259.49   117.8 2258.43   128.4 2261.11   156.5 2262.81   198.7 2259.18
   245.5 2250.57   292.3 2235.61   312.8 2225.92   373.2 2224.31   474.9 2216.97
   491.5 2206.37  500.38 2202.66   512.3  2201.6   518.62202.675   545.4    2219
   616.2 2221.19   644.1 2230.02   660.5 2238.72   684.2  2246.3   732.2 2255.33
   797.3 2263.81   807.8 2271.08   839.5 2287.19   870.4 2297.25   920.8 2308.06
#Mann= 5 ,-1,0
       0      .1       0  138.75     .06       0  500.38    .045       0
   518.6     .06       0  535.18      .1       0
Bank Sta=500.38,518.6
XS Rating Curve= 0 ,0
Exp/Cntr(USF)=0,0
Exp/Cntr=0.3,0.1
